--- LAURELRN5.prj (project) ---

Proj Title=LAURELRN5
Current Plan=p01
Default Exp/Contr=0,0
English Units
Geom File=g01
Flow File=f01
Plan File=p01
BEGIN DESCRIPTION:
----------MODEL BY WOOD PLC 2022----------
AFH study
Randolph County, WV
HEC-RAS Version: RAS 6.2
Vertical Datum: NAVD88
Projection: NAD 1983 StatePlane West Virginia S FIPS 4702 (US Feet)
Terrain: 1-meter LIDAR (FEMA Region III 3DEP collected 2016-2018)
Land Use: 2019 NLCD
Hydrologic Method:
WV SIR2010-5033 regression equations
Additional Model Notes:
None
END DESCRIPTION:
DSS Export Rating Curves= 0
DSS Export Rating Curve Sorted= 0
DSS Export Volume Flow Curves= 0
DXF OffsetX= 0
DXF OffsetY= 0
DXF ScaleX= 0
DXF ScaleY= 0

--- LAURELRN5.p01 (plan) ---

Plan Title=Floodplain
Program Version=6.20
Short Identifier=Floodplain
Geom File=g01
Flow File=f01
Subcritical Flow
K Sum by GR= 0
Std Step Tol= 0.01
Critical Tol= 0.01
Num of Std Step Trials= 20
Max Error Tol= 0.3
Flow Tol Ratio= 0.001
Split Flow NTrial= 30
Split Flow Tol= 0.02
Split Flow Ratio= 0.02
Log Output Level= 0
Friction Slope Method= 1
Unsteady Friction Slope Method= 2
Unsteady Bridges Friction Slope Method= 1
Parabolic Critical Depth
Global Vel Dist= 0 , 0 , 0
Global Log Level= 0
CheckData=True
Encroach Param=-1 ,0,0, 0
Mapping Interval=1HOUR
Computation Time Step Use Courant=        0
Computation Time Step Use Time Series=    0
Computation Time Step Count To Double=0
Computation Time Step Max Doubling=0
Computation Time Step Max Halving=0
Computation Time Step Residence Courant=0
Run HTab= 0
Run UNet= 0
Run Sediment= 0
Run PostProcess= 0
Run WQNet= 0
Run RASMapper=-1
UNET Theta= 0
UNET Theta Warmup= 0
UNET ZTol= 0
UNET ZSATol= 0
UNET MxIter= 0
UNET Max Iter WO Improvement= 0
UNET MaxInSteps= 0
UNET DtIC= 0
UNET DtMin= 0
UNET MaxCRTS= 0
UNET WFStab= 0
UNET SFStab= 0
UNET WFX= 1
UNET SFX= 1
UNET Gravity=32.174
UNET 1D Methodology=Finite Difference
UNET DSS MLevel= 1
UNET Pardiso=0
UNET DZMax Abort= 0
UNET Use Existing IB Tables= 0
UNET Froude Reduction=False
UNET Froude Limit= 0
UNET Froude Power= 0
UNET D1 Cores= 0
UNET WindReference=Eulerian
UNET WindDragFormulation=Hsu (1988)
UNET D2 Coriolis=0
UNET D2 Cores= 0
UNET D2 Theta= 1
UNET D2 Theta Warmup= 1
UNET D2 Z Tol= 0.01
UNET D2 Volume Tol= 0.01
UNET D2 Max Iterations= 20
UNET D2 Equation= 0
UNET D2 RampUpFraction=0.1
UNET D2 TimeSlices= 1
UNET D2 Turbulence Formulation=Non-Conservative (original)
UNET D2 Eddy Viscosity=0.3
UNET D2 Transverse Eddy Viscosity=0.1
UNET D2 Smagorinsky Mixing=0
UNET D2 BCVolumeCheck=0
UNET D2 Cores=0
UNET D2 SolverType=PARDISO (Direct)
UNET D2 Minimum Iterations= 2147483647
UNET D2 Maximum Iterations= 2147483647
UNET D2 Restart Number= 10
UNET D2 Relaxation Coeff=1.3
UNET D2 SOR Precondition Iterations= 10
UNET D2 ILUT Maximum Fill= 8
UNET D2 ILUT Tolerance=1E-08
UNET D1D2 MaxIter= 0
UNET D1D2 ZTol=0.01
UNET D1D2 QTol=0.1
UNET D1D2 MinQTol=1
Write IC File= 0
Write IC File at Fixed DateTime=0
Write IC File at Sim End=0
Echo Input=False
Echo Parameters=False
Echo Output=False
Write Detailed= 0
HDF Write Warmup=0
HDF Write Time Slices=0
HDF Flush=0
HDF Compression= 1
HDF Chunk Size= 1
HDF Spatial Parts= 1
HDF Use Max Rows=0
HDF Fixed Rows= 1
Calibration Method= 0
Calibration Iterations= 20
Calibration Max Change=0.05
Calibration Tolerance=0.2
Calibration Maximum=1.5
Calibration Minimum=0.5
Calibration Optimization Method= 1
WQ AD Non Conservative
WQ ULTIMATE=-1
WQ Max Comp Step=1HOUR
WQ Output Interval=15MIN
WQ Output Selected Increments= 0
WQ Output face flow=0
WQ Output face velocity=0
WQ Output face area=0
WQ Output face dispersion=0
WQ Output cell volume=0
WQ Output cell surface area=0
WQ Output cell continuity=0
WQ Output cumulative cell continuity=0
WQ Output face conc=0
WQ Output face dconc_dx=0
WQ Output face courant=0
WQ Output face peclet=0
WQ Output face adv mass=0
WQ Output face disp mass=0
WQ Output cell mass=0
WQ Output cell source sink temp=0
WQ Output nsm pathways=0
WQ Output nsm derived pathways=0
WQ Create Restart=0
WQ Fixed Restart=0
WQ System Summary=0
WQ Write To DSS=0
Sorting and Armoring Iterations= 10
XS Update Threshold= 0.02
Bed Roughness Predictor= 0
Hydraulics Update Threshold= 0.02
Energy Slope Method= 1
Volume Change Method= 1
Sediment Retention Method= 0
Sediment TS Multiplier= 1
Warm Up Method= 0
XS Weighting Method= 0
Number of US Weighted Cross Sections= 1
Number of DS Weighted Cross Sections= 1
Upstream XS Weight=0
Main XS Weight=1
Downstream XS Weight=0
Number of DS XS's Weighted with US Boundary= 1
Upstream Boundary Weight= 1
Weight of XSs Associated with US Boundary= 0
Number of US XS's Weighted with DS Boundary= 1
Downstream Boundary Weight= 0.5
Weight of XSs Associated with DS Boundary= 0.5
Percentile Method= 0
Sediment Output Level= 3
Mass or Volume Output= 0
Output Increment Type= 1
Profile and TS Output Increment= 1
Transport Output Increment 1
XS Output Flag= 0
XS Output Increment= 10
Read HDF5 Sediment Hotstart= 0
Sediment Hotstart Type= 0
Write Gradation File= 0
Read Gradation Hotstart= 0
Write HDF5 File= 1
Write Binary Output= 1
Write DSS Sediment File= 0
DSS Sediment Output Type= 1
SV Curve= 0
Specific Gage Flag= 0
Subcell Erosion Methods= 0
Subcell Deposition Methods= 0
Advection Scheme= 1
Matrix Solver= 0
Implicit Weighting Factor= 1
Maximum Outer Loop Convergence Iterations= 5
Convergence Maximum Absolute= 0.001
Convergence RMSE= 0.0001
Grain Fractions Max Abs Error= 0.001
Max Subgrid Regions= 1
Max Subgrid Length Scale= 3.402823E+38
Initial Layer Thickness= 3.402823E+38
Min Layer Thickness= 3.402823E+38
Max Layer Thickness= 3.402823E+38
Number of Layers= 5

--- LAURELRN5.f01 (steady flow) ---

Flow Title=Flow
Program Version=6.20
Number of Profiles= 1
Profile Names=P100yr
River Rch & RM=LAURELRN5,Main,7389
     357
River Rch & RM=LAURELRN5,Main,4522
     443
River Rch & RM=LAURELRN5,Main,2107
     501
Boundary for River Rch & Prof#=LAURELRN5,Main            , 1
Up Type= 0
Dn Type= 3
Dn Slope=0.03677
DSS Import GetInterval= 0
DSS Import GetPeak= 0
DSS Import FillOption= 0

--- LAURELRN5.g01 (geometry) ---

Geom Title=Geometry
Program Version=6.20

River Reach=LAURELRN5       ,Main
Reach XY= 30
2270652.47614156617237.973707289     2270453.715      617215.162
2270299.28800003616943.8079999982270217.52700001 616896.74500002
2270178.71500003616819.7629999972269981.26500003616797.566000015
2269993.99300005616619.7630000112269832.88200004616431.568000019
2269838.04190788616348.5183870052269595.39614797615905.112891704
2269638.85663989615662.7130749822269583.56172204615591.154803678
2269529.59712626615598.5595116472269533.33799998      615377.044
2269457.47699998615299.4790000022269413.20600002615183.159999996
2269449.66399999615045.1390000132269563.53900003614896.285999998
2269475.91200003614754.7810000182269324.98100004614647.886000022
2269180.56699999614427.9520000222269196.62700002614129.342000008
2268920.58400002613888.4550000132268932.26699999613636.936000004
2268762.12800001612774.9570000172268644.94099998612406.033000022
2268453.10000001612046.658000007     2268287.302611931.207000002
2268118.89900005611906.900999993     2267531.366      611725.396

Type RM Length L Ch R = 1 ,7389    ,128.8,125.6,122.7
XS GIS Cut Line= 4
2270729.84294779617187.2199571922270668.79237014617208.198171757
 2270626.0587305617279.2367447932270597.02340145617370.457773913
#Sta/Elev= 30
       0 2499.39    10.2 2493.98    31.2 2484.28    52.5 2473.55      61 2471.12
    68.6 2468.07    71.5 2467.89    79.7  2468.9    83.2 2467.86    84.4 2467.02
      89 2462.06   92.792459.778    98.4 2458.51  103.682459.779   107.7 2461.71
   112.3 2462.34   121.7 2462.17   135.7 2461.09   141.5 2462.46   145.1    2464
   149.5 2466.63   153.7 2468.19   157.9 2469.03   166.4 2469.65   174.7 2471.65
   191.5 2477.93   204.6 2485.24   216.7 2489.96   229.3 2493.55   243.2 2499.83
#Mann= 3, -1 ,  0
       0     0.1       0   92.79   0.045       0  103.68     0.1       0
Bank Sta=92.79,103.68
XS Rating Curve= 0 ,0
Exp/Cntr=0.3,0.1

Type RM Length L Ch R = 1 ,7264    ,108.7,116.3,120.4
XS GIS Cut Line= 4
2270559.34993684617114.8621226882270532.98310377617199.860466144
2270532.98310377617246.696288048 2270496.9021743617316.082690869
#Sta/Elev= 30
       0 2478.96     2.4 2477.48     6.6 2474.33     7.6 2473.84    20.4 2469.01
    26.8 2468.07    31.7 2467.67    35.9 2466.44    40.1 2465.64    44.3 2465.73
    52.7 2466.46    56.9 2466.01    61.9 2464.73    73.6 2463.99      82 2463.01
    86.2 2462.26    94.3 2457.87   102.3 2457.38  107.462456.003   110.3 2455.27
   114.3 2455.18  123.352456.001   126.3 2456.48   138.3 2460.47   147.6 2464.84
   153.1 2467.12   172.3 2474.18   197.2 2488.03   201.7 2490.79     214 2497.23
#Mann= 3, -1 ,  0
       0     0.1       0  107.46   0.045       0  123.35     0.1       0
Bank Sta=107.46,123.35
XS Rating Curve= 0 ,0
Exp/Cntr(USF)=0,0
Exp/Cntr=0.3,0.1

Type RM Length L Ch R = 1 ,7148    ,120.6,123.4,125.2
XS GIS Cut Line= 4
2270499.13530871 617109.773679692270451.60946613617169.002305347
2270419.56456268617200.4215581172270364.61257078 617262.67021785
#Sta/Elev= 30
       0 2466.92     4.4 2465.03     9.5 2463.39    19.8 2461.01    24.9  2460.8
    35.1 2462.07    40.3 2462.07    50.5  2460.8    61.4 2458.12    65.9 2457.62
    76.2 2457.31    86.4 2456.37      92 2454.81   98.282451.796   101.1 2451.33
   108.8 2450.89   110.5 2451.13  112.082451.795   114.4 2453.14     132 2466.92
     138 2470.79   140.8 2472.89   150.1 2480.99   156.2  2485.3   168.2 2494.92
   174.8    2499   180.4 2503.06   188.9 2508.65   200.3 2515.21   203.9 2517.01
#Mann= 3, -1 ,  0
       0     0.1       0   98.28   0.045       0  112.08     0.1       0
Bank Sta=98.28,112.08
XS Rating Curve= 0 ,0
Exp/Cntr=0.3,0.1

Type RM Length L Ch R = 1 ,7024    ,121.3,119.6,119.2
XS GIS Cut Line= 4
2270473.62540122617039.2002609072270387.83217755617075.207801337
2270355.94679353617089.484838955 2270303.5976556617136.123161838
#Sta/Elev= 30
       0 2472.55    14.6  2465.2    23.3 2462.14    27.6 2460.94    33.2 2460.17
      45 2460.25    49.3 2459.86    53.6 2458.74    60.7 2455.77    63.7 2455.13
    66.6 2454.89      79 2455.91    85.1 2455.95    88.2 2455.32   101.4  2450.9
   105.8 2448.77  108.622447.133   110.2 2446.33   114.6  2446.1  118.932447.136
   123.3 2449.15   124.5    2450   138.4  2460.4   149.1  2468.7   154.5 2471.57
   159.8 2475.13   163.6  2477.4   175.9 2483.33     192 2490.43   198.1 2493.71
#Mann= 3, -1 ,  0
       0     0.1       0  108.62   0.045       0  118.93     0.1       0
Bank Sta=108.62,118.93
XS Rating Curve= 0 ,0
Exp/Cntr(USF)=0,0
Exp/Cntr=0.3,0.1

Type RM Length L Ch R = 1 ,6905    ,114.5,108.5,104.2
XS GIS Cut Line= 4
2270412.35654552616902.0101615212270358.82759227616949.990508146
2270310.42612211616980.4934184912270244.24425684617043.283082019
#Sta/Elev= 30
       0 2476.06      11 2470.09    19.4 2466.24    28.7 2461.42    34.7 2458.88
      42 2456.27    52.7 2453.69    58.7 2451.78    64.7 2450.72    79.7 2448.99
    87.7 2449.06    93.9 2449.72    96.4 2449.25    98.7 2448.29   103.4 2443.53
   107.9 2441.65   112.8 2440.89   116.7 2440.79   122.42441.651   128.3  2444.3
   132.2 2446.58   137.7 2448.91   141.7  2450.4   154.3  2453.8   159.5 2455.66
   165.1  2458.4   190.6  2474.3   198.4 2478.38   213.2 2487.02   220.3 2490.39
#Mann= 3, -1 ,  0
       0     0.1       0   107.9   0.045       0   122.4     0.1       0
Bank Sta=107.9,122.4
XS Rating Curve= 0 ,0
Exp/Cntr=0.3,0.1

Type RM Length L Ch R = 1 ,6796    ,133.1,133.3,130.7
XS GIS Cut Line= 4
2270339.01882131616800.5569453572270245.46689898616889.274339606
2270236.44666662616922.2328809452270200.20726203616970.113041712
#Sta/Elev= 30
       0 2484.43     3.9 2482.03    13.8 2477.21      26 2467.14    42.5 2455.02
    47.7 2452.18    53.5 2449.85    64.6 2448.73    70.4 2447.31      76 2446.79
    81.1 2447.22    88.1 2448.97    92.1 2449.41    98.7 2447.84   111.4 2446.35
   124.1 2446.68   128.8 2445.19   136.4 2437.02  140.472434.669   141.3 2434.27
   146.2 2433.86   149.6 2433.87  154.042434.668   157.9 2436.67   166.8 2442.43
   176.9 2447.83   191.9 2458.88   199.7 2464.11   209.9 2471.58   223.1 2479.14
#Mann= 3, -1 ,  0
       0     0.1       0  140.47   0.045       0  154.04     0.1       0
Bank Sta=140.47,154.04
XS Rating Curve= 0 ,0
Exp/Cntr(USF)=0,0
Exp/Cntr=0.3,0.1

Type RM Length L Ch R = 1 ,6663    ,134.8,131.6,126.5
XS GIS Cut Line= 4
2270232.93752686616731.1614349922270167.88585637616791.439666977
2270150.39831905616835.1212994642270115.46263689616931.902705055
#Sta/Elev= 30
       0 2477.87     8.9  2473.2    22.9 2464.18    30.3 2458.81    39.2 2453.26
    52.9 2446.56    58.6 2444.44    61.8 2443.62    69.9 2443.17    79.5  2444.1
    82.8 2443.77    85.4 2442.91    90.6 2437.71    94.9 2431.27      99 2426.46
  100.512425.989   103.5 2425.34   108.3 2425.23  120.062425.989     125 2426.88
   129.3 2428.45   133.6 2429.52   137.9 2431.39   146.4 2437.21   154.9  2440.7
   167.2 2447.69   173.5 2451.61   193.2 2464.97   214.1 2474.95   238.6 2487.47
#Mann= 3, -1 ,  0
       0     0.1       0  100.51   0.045       0  120.06     0.1       0
Bank Sta=100.51,120.06
XS Rating Curve= 0 ,0
Exp/Cntr=0.3,0.1

Type RM Length L Ch R = 1 ,6531    ,90.9,110,116.1
XS GIS Cut Line= 4
2270129.24505253616720.8823724152270030.53960728616786.686002586
2270032.88973693616831.3384659172270021.13908868616890.091707141
#Sta/Elev= 30
       0 2440.93     9.6 2437.08    15.4 2436.53    22.2 2437.08    34.9 2440.01
    38.5 2440.45    49.4 2438.63    58.7 2439.02    67.3 2438.68    73.1 2439.96
    78.9 2440.62    94.3 2439.98   101.5 2437.93   118.8 2430.28   122.6 2428.22
   129.1 2423.83  136.782421.891   141.2  2421.2   145.2 2421.18  153.712421.889
   157.2 2423.66   161.2 2427.63   165.2 2432.48   173.4 2439.59   177.5 2444.51
   185.9 2456.57   193.8 2465.47   201.9 2473.49   206.3 2477.09   223.3 2487.01
#Mann= 3, -1 ,  0
       0     0.1       0  136.78   0.045       0  153.71     0.1       0
Bank Sta=136.78,153.71
XS Rating Curve= 0 ,0
Exp/Cntr(USF)=0,0
Exp/Cntr=0.3,0.1

Type RM Length L Ch R = 1 ,6421    ,142.2,137.4,134.5
XS GIS Cut Line= 4
2270093.21244144616683.6378041072270021.43501726616749.035626519
2269960.76344829616746.5177489372269869.19436213616765.754828212
#Sta/Elev= 30
       0 2433.91     6.8 2433.24    10.3 2433.29    14.2 2433.67      26 2435.71
    39.3 2435.23    72.6 2437.45    81.1 2435.93    89.6 2435.83    98.6 2434.07
   106.4 2430.31   114.4 2425.21   122.4 2420.66   126.4 2419.56   134.4 2419.17
  138.872417.778   142.4 2416.94   146.4 2416.81  150.972417.778   154.4 2419.95
   162.5  2431.6   166.6 2436.56   170.7 2440.33   175.8 2444.42     183 2449.96
     187  2452.6   199.3 2457.16   211.6 2461.07   219.7 2464.04   251.4 2473.58
#Mann= 3, -1 ,  0
       0     0.1       0  138.87   0.045       0  150.97     0.1       0
Bank Sta=138.87,150.97
XS Rating Curve= 0 ,0
Exp/Cntr=0.3,0.1

Type RM Length L Ch R = 1 ,6284    ,111.4,108.1,106
XS GIS Cut Line= 4
2270081.23067413616566.0974241892270008.89368354616606.549030772
2269966.53847194616627.488685945 2269907.0508152616682.217330145
#Sta/Elev= 30
       0 2471.22     8.9 2464.26      15  2460.1    22.7 2454.19    38.3 2443.34
    42.5 2440.74      47  2438.5    56.2 2435.56    60.8 2432.66    63.7 2431.62
    67.7 2431.01    74.5 2431.27    79.1 2429.32    88.8 2417.93   92.482414.333
    97.1 2413.34   101.5 2413.35  107.182414.338   110.5 2414.87   119.4 2415.08
   123.8 2416.86   128.3 2419.29   132.6 2420.65   138.8 2421.64     150 2422.39
     167 2427.55   182.3 2428.63   185.8 2429.22   206.6 2435.98     211 2438.01
#Mann= 3, -1 ,  0
       0     0.1       0   92.48   0.045       0  107.18     0.1       0
Bank Sta=92.48,107.18
XS Rating Curve= 0 ,0
Exp/Cntr(USF)=0,0
Exp/Cntr=0.3,0.1

Type RM Length L Ch R = 1 ,6176    ,110.2,112.3,114.3
XS GIS Cut Line= 4
2270026.99579362616485.4565626622269939.23609953616515.438524538
2269901.85340164616555.1748966782269829.20171499616613.670106653
#Sta/Elev= 30
       0 2476.95     7.2 2474.03    17.8 2468.92    36.8 2458.72    45.3 2451.27
    52.4 2445.89      61 2438.23    83.9 2420.77    87.5 2419.58    96.1 2419.87
      99 2419.15   106.1 2413.73   108.9 2412.32  111.982411.637   126.4 2410.87
  131.792411.636   139.1 2414.93   149.9 2417.36   158.5 2418.58   169.6 2423.09
   172.7 2423.85   185.4 2425.49   195.7 2424.96   201.1 2426.04   205.9 2426.52
   215.3  2428.9   220.7 2429.52   226.5 2430.71   231.6 2432.71   240.6 2438.59
#Mann= 3, -1 ,  0
       0     0.1       0  111.98   0.045       0  131.79     0.1       0
Bank Sta=111.98,131.79
XS Rating Curve= 0 ,0
Exp/Cntr=0.3,0.1

Type RM Length L Ch R = 1 ,6063    ,134.5,136.3,136.5
XS GIS Cut Line= 4
2269983.12782666616395.3897561482269873.67053826616433.990635633
2269829.75891477616462.522196773 2269792.3277259616495.906770626
#Sta/Elev= 30
       0 2474.74    16.3 2464.22    24.3 2457.43    32.8 2451.12    41.3 2443.55
    53.5  2434.2      71 2422.54    75.2 2420.21    91.5  2415.2    96.4 2414.37
   100.7  2414.5   113.4 2416.12   117.8 2414.56   122.6 2410.97   125.2 2409.94
   127.4 2409.33   133.9 2409.36  141.012408.021   151.2 2407.03  156.062408.022
   165.7 2409.78   170.6 2413.02   179.9 2420.98   182.8 2423.01   186.6 2424.93
     192 2425.93   197.4 2427.95   208.1 2436.45   213.4 2439.01   218.6 2440.79
#Mann= 3, -1 ,  0
       0     0.1       0  141.01   0.045       0  156.06     0.1       0
Bank Sta=141.01,156.06
XS Rating Curve= 0 ,0
Exp/Cntr(USF)=0,0
Exp/Cntr=0.3,0.1

Type RM Length L Ch R = 1 ,5927    ,85.1,85.4,85.7
XS GIS Cut Line= 4
2269926.60174355616298.7914447132269840.75492842616316.137284503
 2269786.1064902616351.1296842632269728.66302611 616381.91392846
#Sta/Elev= 30
       0 2469.33    14.7 2460.59      31 2451.65    43.3 2445.83    51.6 2441.25
      55 2439.15    63.7 2432.44    67.8 2430.53      72 2429.41    75.4  2426.9
    78.8  2423.4    84.1 2416.49    88.3 2410.38    89.5 2409.03      93 2407.29
    97.8 2406.75   105.6  2403.2   107.3 2402.81   111.8  2402.6   118.62403.186
   126.3 2403.89   129.3  2404.6   140.5 2409.77     150 2411.93   163.7 2419.24
   170.2  2421.2   177.4 2421.96   182.2 2421.58     191 2421.47   217.6 2421.92
#Mann= 3, -1 ,  0
       0     0.1       0   105.6   0.045       0   118.6     0.1       0
Bank Sta=105.6,118.6
XS Rating Curve= 0 ,0
Exp/Cntr=0.3,0.1

Type RM Length L Ch R = 1 ,5842    ,133.2,134.4,135.4
XS GIS Cut Line= 4
2269888.26887252  616232.4087121 2269801.3140755 616242.98429552
2269735.91455013616281.6496860642269687.34406815616316.342887474
#Sta/Elev= 30
       0 2462.53    28.3 2446.42    36.4 2440.38    40.3 2437.17    52.5 2426.12
    56.5 2422.76    65.4 2415.75      69 2413.39    72.6 2412.09    93.6 2408.14
    98.2 2408.02   102.9  2408.5   104.6 2408.32   107.5 2407.48   112.2 2403.33
   113.4 2402.61   116.3 2401.41  117.922401.064   121.4 2400.36   126.1 2400.14
   130.9 2400.26     1342401.063     154 2409.09   165.9 2415.53   168.2 2416.58
   169.6 2416.93   176.5 2417.91     186 2417.86   192.7 2418.41   223.3 2418.52
#Mann= 3, -1 ,  0
       0     0.1       0  117.92   0.045       0     134     0.1       0
Bank Sta=117.92,134
XS Rating Curve= 0 ,0
Exp/Cntr(USF)=0,0
Exp/Cntr=0.3,0.1

Type RM Length L Ch R = 1 ,5707    ,120.2,120.5,120.1
XS GIS Cut Line= 4
 2269821.1032679616116.600117817 2269745.1110577616126.826775027
2269675.08884728616155.8833249442269614.34444503616187.918532959
#Sta/Elev= 30
       0 2446.44       9 2443.29    15.6 2440.39    33.2 2429.83    40.5 2424.63
    45.3 2419.95    49.4 2416.75    57.4 2411.03    61.8 2408.73    65.5  2407.5
      76 2407.18      82 2406.55    85.3 2404.93    99.3  2399.8  103.72 2397.67
     108 2396.94   112.3 2396.86   116.7 2397.09     119 2397.64   125.1 2399.87
     135 2405.71   142.7 2407.94   151.3  2412.6   155.8 2413.96   160.3 2414.65
   173.9 2415.41   187.4 2415.68     210 2417.23   217.8 2416.94   221.2 2417.47
#Mann= 3, -1 ,  0
       0     0.1       0  103.72   0.045       0     119     0.1       0
Bank Sta=103.72,119
XS Rating Curve= 0 ,0
Exp/Cntr=0.3,0.1

Type RM Length L Ch R = 1 ,5587    ,124.4,124.3,123.6
XS GIS Cut Line= 4
2269785.47385409616023.6220727192269699.81162839616015.484161277
2269618.00420284616051.0339849452269557.61233372616065.168252186
#Sta/Elev= 30
       0 2432.17    17.4 2420.14    25.4 2415.91    33.4 2410.43    41.5 2406.77
    53.5 2405.16    57.6  2403.2    61.6 2402.11    65.6 2402.05    73.6 2402.94
    85.7  2400.4    98.7 2399.06   103.1 2398.11   108.3 2395.39   111.8 2394.49
   116.2 2394.29  122.282395.406   124.9 2396.15   129.3 2396.14   138.7 2395.07
     157 2397.81   159.8 2398.39   164.2 2400.19   177.1 2407.13   181.2  2408.2
   197.7 2408.97     210 2413.84   214.1 2415.91   225.2 2422.68   237.3  2430.9
#Mann= 3, -1 ,  0
       0     0.1       0   108.3   0.045       0  122.28     0.1       0
Bank Sta=108.3,122.28
XS Rating Curve= 0 ,0
Exp/Cntr(USF)=0,0
Exp/Cntr=0.3,0.1

Type RM Length L Ch R = 1 ,5462    ,135.7,139.1,139.5
XS GIS Cut Line= 4
2269752.57339083615906.0210352232269630.87577935615911.968220501
  2269575.537208615935.5430570772269490.24942978615977.701545417
#Sta/Elev= 30
       0 2420.52    16.4 2411.76    32.4 2401.69    40.4 2398.25    48.5 2397.52
    56.8 2398.57    68.5 2398.79   100.5  2401.7   108.5 2401.23   120.5 2401.55
   124.8 2400.17   129.1 2395.42   130.9 2394.32   133.5 2393.48  140.812393.749
   149.1 2393.65   159.6 2394.27   167.5 2392.96   170.6 2394.05   182.7 2400.82
   188.7 2405.51   194.7 2411.33   206.6  2425.2   209.6 2427.55   212.6 2429.04
     217 2430.31   234.8 2433.05   257.1 2434.74   266.1  2433.9   277.1 2435.77
#Mann= 3, -1 ,  0
       0     0.1       0  140.81   0.045       0   149.1     0.1       0
Bank Sta=140.81,149.1
XS Rating Curve= 0 ,0
Exp/Cntr=0.3,0.1

Type RM Length L Ch R = 1 ,5323    ,94.3,93.4,93.2
XS GIS Cut Line= 3
2269764.85447625615793.6974586722269540.85017301615785.465741619
 2269478.3182803615793.206806859
#Sta/Elev= 30
       0 2420.38     8.9  2414.5    16.7 2408.53    20.7 2406.12    40.7 2394.81
    44.7 2393.69    52.7 2393.13    64.7 2395.07    80.7 2395.35    88.7 2397.09
   104.8 2397.56   108.8 2397.37   112.8 2396.46   124.7 2391.15   128.8 2389.95
   147.9 2388.98   152.8 2388.61   162.82388.981   172.8 2389.83   180.8 2389.37
   196.8 2390.08   208.8 2392.15   216.8 2392.61   220.8 2393.73   234.5 2400.21
     241 2404.01   252.9 2411.97   265.1  2421.5   277.2 2427.59   287.2 2431.59
#Mann= 3, -1 ,  0
       0     0.1       0   147.9   0.045       0   162.8     0.1       0
#XS Ineff= 2 , 0
                          173.36         2408.43
Permanent Ineff=
       F       F
Bank Sta=147.9,162.8
XS Rating Curve= 0 ,0
Exp/Cntr(USF)=0,0
Exp/Cntr=0.3,0.1

Type RM Length L Ch R = 1 ,5230    ,70.3,67.3,64.6
XS GIS Cut Line= 4
2269749.32014326615704.8592048572269658.29161694615701.224252043
 2269560.4984208615704.8774461522269471.68421066615721.559479311
#Sta/Elev= 30
       0 2405.07     9.2 2400.78    13.2 2399.35    21.2 2397.68    29.2 2394.29
    33.2  2393.2    49.2 2392.46    57.2 2393.68    69.2 2392.93    81.2 2393.74
    85.2 2392.66    89.2 2390.01    93.2  2388.2    97.2 2387.73   105.2 2387.26
   112.4 2387.74   121.2 2387.45   129.2  2388.1   145.3  2388.2   153.3 2387.36
   157.3 2386.23   165.3  2386.1   177.3 2384.19   206.6 2390.16   217.8 2394.21
   225.9 2398.52   244.1 2412.04   250.3  2416.1   259.1  2419.9   279.3 2425.71
#Mann= 3, -1 ,  0
       0     0.1       0    97.2   0.045       0   112.4     0.1       0
#XS Ineff= 2 , 0
                          137.76         2401.72
Permanent Ineff=
       F       F
Bank Sta=97.2,112.4
XS Rating Curve= 0 ,0
Exp/Cntr(USF)=0,0
Exp/Cntr=0.3,0.1

Type RM Length L Ch R = 1 ,5163    ,156.1,166.3,164.3
XS GIS Cut Line= 4
2269754.13016491615623.6860822752269643.79294586615629.963306983
 2269545.7918303615676.5187407072269471.94569571615685.666836984
#Sta/Elev= 30
       0 2418.48    14.6 2407.34      30 2396.46      38 2392.57      50 2390.16
      58 2389.79    82.1 2391.77    94.1 2389.88   106.1 2390.05   110.1 2389.45
   118.6 2384.74   124.7 2382.07   127.8 2381.42  137.392382.062   141.1  2382.3
   149.9 2384.18   154.4  2384.4   163.2 2383.69   172.1  2383.8   181.7 2384.74
   196.7 2383.97   201.9 2384.15   208.7 2386.35   216.4 2388.09   224.7 2388.66
   228.7 2390.23   232.7 2392.75   252.9 2409.13   256.9 2411.56   293.4 2422.45
#Mann= 3, -1 ,  0
       0     0.1       0   124.7   0.045       0  137.39     0.1       0
#XS Ineff= 2 , 0
                           154.1         2392.08
Permanent Ineff=
       F       F
Bank Sta=124.7,137.39
XS Rating Curve= 0 ,0
Exp/Cntr=0.3,0.1

Type RM Length L Ch R = 1 ,4996    ,102.8,102.9,103
XS GIS Cut Line= 3
2269699.93662722615526.3550518072269557.76829043615561.171787348
2269452.59273515615562.622484662
#Sta/Elev= 30
       0 2400.74     3.9 2398.44     8.8 2396.73    16.2  2392.9    20.3 2391.26
    24.5 2390.54    28.6 2390.85    40.9 2394.15    53.3 2394.88    62.3 2394.83
    69.8  2393.9    82.1 2391.01    94.5 2386.43   106.8 2382.86   110.9 2382.11
   127.8 2382.39   139.8 2380.79     156 2380.25  169.17 2377.72   176.4 2376.81
     180 2376.82  182.03 2377.72     184 2378.56     188 2382.23     196 2390.94
   207.1 2401.12     212 2405.02     216 2406.96     220 2407.88   251.6 2413.87
#Mann= 3, -1 ,  0
       0     0.1       0  169.17   0.045       0  182.03     0.1       0
Bank Sta=169.17,182.03
XS Rating Curve= 0 ,0
Exp/Cntr(USF)=0,0
Exp/Cntr=0.3,0.1

Type RM Length L Ch R = 1 ,4893    ,104.5,100.3,96.5
XS GIS Cut Line= 4
2269687.28748458615436.0467159092269554.01793272615459.116120114
2269505.80169492615458.5169890752269436.94803325615460.451697569
#Sta/Elev= 30
       0 2405.35     3.2 2404.28    19.4 2400.64    43.8 2394.31    48.7 2394.53
      60  2396.5    76.3 2400.95    84.3 2402.46   100.6 2403.06   107.5 2402.46
   112.8 2400.64   116.8 2398.61   120.9 2395.05     129 2385.61   133.1 2381.35
   141.1 2376.12   145.1 2374.19   147.1 2373.81   157.1 2372.79   161.1 2372.91
  167.53 2373.81   173.1  2374.6   177.1 2376.18   185.1 2383.78   189.1 2386.69
   201.1 2397.59   205.1 2400.64   213.1 2402.85   241.1    2408   252.4 2410.48
#Mann= 3, -1 ,  0
       0     0.1       0   147.1   0.045       0  167.53     0.1       0
Bank Sta=147.1,167.53
XS Rating Curve= 0 ,0
Exp/Cntr=0.3,0.1

Type RM Length L Ch R = 1 ,4793    ,144.9,146.8,149.7
XS GIS Cut Line= 4
2269604.63662269615314.332409377 2269534.2502397 615352.40450969
2269500.21405137615381.8513017842269448.67512871615412.221369661
#Sta/Elev= 30
       0  2397.7     5.1 2395.83    27.8 2390.24    32.4  2389.7    39.6 2389.83
    43.8 2390.54      48 2391.78    50.5 2392.05    56.4 2391.26    64.2 2389.54
    81.2 2381.16      82 2380.35    87.7 2372.61   90.072371.453    93.4 2370.28
    96.2 2370.38  100.532371.452   110.4 2376.28   118.9 2376.35   124.6 2379.09
   127.5 2381.32   129.7 2383.55   136.3    2392   139.2 2395.37   143.6 2398.53
   147.9 2400.69   159.6 2404.89   168.4 2407.49   178.9 2409.92   184.9 2410.61
#Mann= 3, -1 ,  0
       0     0.1       0   90.07   0.045       0  100.53     0.1       0
Bank Sta=90.07,100.53
XS Rating Curve= 0 ,0
Exp/Cntr(USF)=0,0
Exp/Cntr=0.3,0.1

Type RM Length L Ch R = 1 ,4646    ,120.2,124.5,130.4
XS GIS Cut Line= 4
2269541.06215378615216.8288139472269461.71994926615238.432155859
 2269399.7972998615262.225895118 2269344.5592198615317.228216475
#Sta/Elev= 30
       0 2404.77    13.4 2402.51    34.1 2396.55    38.2  2396.2    46.5 2396.59
    59.7 2394.57    63.1 2393.26    67.2 2390.76      76 2383.48    79.7 2379.75
    83.9  2374.2    88.2 2372.32    96.7  2369.8  104.072366.854   105.3 2366.33
   109.6 2365.66   113.9 2365.68   118.2 2366.49  118.622366.853   122.5  2370.5
   126.7 2375.03     131 2375.66   138.2 2375.69   143.9 2377.14   169.8 2378.51
   181.5 2381.54   198.1 2391.83   210.1 2401.07   220.8 2408.82   226.5 2411.64
#Mann= 3, -1 ,  0
       0     0.1       0  104.07   0.045       0  118.62     0.1       0
Bank Sta=104.07,118.62
XS Rating Curve= 0 ,0
Exp/Cntr=0.3,0.1

Type RM Length L Ch R = 1 ,4522    ,125.3,130.7,135.9
XS GIS Cut Line= 4
2269533.27315732615181.2778541682269450.36580581615134.275261188
2269382.47317151615121.2189853612269279.32859247 615115.99647503
#Sta/Elev= 30
       0 2400.65    18.5 2393.09    28.9 2389.79      38  2387.9    47.2 2386.94
    56.4 2384.53      61 2384.25    65.6 2383.17    94.8 2370.67   101.6 2369.05
   109.8    2368   113.8 2366.78  117.692364.647     122 2363.82  138.832364.648
   142.5 2367.15   146.4 2367.26   154.6 2366.38   158.6 2367.52   162.7 2370.53
   166.7 2371.35   170.7  2370.7   189.5 2371.79   218.8 2375.51   227.7 2377.66
   234.8 2380.17   239.1 2382.32   242.8 2384.99   259.6 2399.49   267.7 2405.02
#Mann= 3, -1 ,  0
       0     0.1       0  117.69   0.045       0  138.83     0.1       0
#XS Ineff= 2 , 0
                          145.21         2371.78
Permanent Ineff=
       F       F
Bank Sta=117.69,138.83
XS Rating Curve= 0 ,0
Exp/Cntr(USF)=0,0
Exp/Cntr=0.3,0.1

Type RM Length L Ch R = 1 ,4391    ,118.4,115.9,110.8
XS GIS Cut Line= 4
2269576.38611348615081.4175740222269521.45367555615058.074888988
2269437.19169693614975.5703325662269353.16648082614950.112206921
#Sta/Elev= 30
       0 2400.95    30.8 2383.83      43 2376.11      48  2374.7    52.2 2372.86
    56.7 2369.66    61.5 2366.87    67.1 2365.52    86.7 2365.05    95.1 2364.15
   103.7 2362.58   112.4 2362.28  119.25 2360.49   123.1 2359.74   128.7  2359.6
   135.3 2360.49   145.4 2363.44   154.6 2362.56   173.4 2363.56   177.6  2364.1
   182.9 2365.63     187 2366.35   191.2 2366.09   199.6 2364.44   203.8 2365.53
   215.6 2370.66   220.5 2373.89   249.7 2396.96   257.3 2403.26   265.4 2408.74
#Mann= 3, -1 ,  0
       0     0.1       0  119.25   0.045       0   135.3     0.1       0
#XS Ineff= 2 , 0
          109.25  2371.1  145.87         2371.01
Permanent Ineff=
       F       F
Bank Sta=119.25,135.3
XS Rating Curve= 0 ,0
Exp/Cntr=0.3,0.1

Type RM Length L Ch R = 1 ,4275    ,117.5,110.5,98.2
XS GIS Cut Line= 4
2269633.81257054614974.7097999782269572.42130879614939.493107188
2269478.51809857614896.2372182012269365.67941135614914.238541484
#Sta/Elev= 30
       0 2418.91    15.7 2409.37    25.8 2402.44    34.6 2394.44    43.4 2384.87
    52.1 2376.72    61.8 2369.71    66.8 2367.12    70.8 2363.09    75.7 2356.59
   78.442355.552    93.8 2354.85   100.12355.554   106.3  2358.5   110.7 2359.34
     133 2360.45   154.7 2359.91   163.5 2361.13   167.9 2360.91   172.3 2360.47
   180.6 2358.22   187.5  2357.6   196.8 2359.09   221.1 2360.49   225.1 2362.04
   241.3 2374.64   249.4 2379.78   257.5  2387.3   265.6 2392.15   288.4 2409.35
#Mann= 3, -1 ,  0
       0     0.1       0   78.44   0.045       0   100.1     0.1       0
Bank Sta=78.44,100.1
XS Rating Curve= 0 ,0
Exp/Cntr(USF)=0,0
Exp/Cntr=0.3,0.1

Type RM Length L Ch R = 1 ,4165    ,128.7,123.6,120.6
XS GIS Cut Line= 4
2269613.40603931614793.9416988252269537.70171515 614827.73534088
2269471.40175323614866.585502192 2269366.1053047614892.052757366
#Sta/Elev= 30
       0 2429.85     5.7 2427.59    10.1 2424.12    18.5 2416.24    27.6 2408.73
    36.4 2399.44    45.2 2393.18    49.5 2389.26    60.9 2378.11      67 2371.53
    79.1 2356.42   87.862352.116    93.8 2350.89  100.782352.117   112.5 2356.56
   141.1 2358.48   149.6 2360.48   154.2 2360.73   158.9 2360.09   171.2 2356.83
   175.4 2356.56   183.6 2357.74   200.1 2358.88   204.2 2360.05   216.6 2370.36
   241.3 2388.18   249.5 2394.78   253.6 2396.94   261.8 2404.91   268.1 2409.31
#Mann= 3, -1 ,  0
       0     0.1       0   87.86   0.045       0  100.78     0.1       0
Bank Sta=87.86,100.78
XS Rating Curve= 0 ,0
Exp/Cntr=0.3,0.1

Type RM Length L Ch R = 1 ,4041    ,115.8,117.6,118.4
XS GIS Cut Line= 4
2269592.06373798  614680.81307982269462.15379349614721.940348657
 2269427.1666803614778.2875859012269344.94379295614825.123407805
#Sta/Elev= 30
       0 2452.51     8.3  2447.7    16.1  2441.9    35.3 2429.38    62.8  2410.5
    71.2 2405.98      94 2387.49   104.8 2379.86   113.2 2373.04   118.1 2370.47
   121.6 2367.95   140.1 2349.43  143.992348.292   154.2 2347.48  161.612348.293
   163.6 2348.94   169.1  2352.9     173 2354.38   193.1 2351.88   200.7 2352.01
     206 2352.86   212.8 2355.19   215.2 2355.49   219.8 2354.94   230.4 2357.03
   233.7 2358.76   261.3 2379.23   273.1 2386.69   289.2 2398.09   297.2 2402.98
#Mann= 3, -1 ,  0
       0     0.1       0  143.99   0.045       0  161.61     0.1       0
Bank Sta=143.99,161.61
XS Rating Curve= 0 ,0
Exp/Cntr(USF)=0,0
Exp/Cntr=0.3,0.1

Type RM Length L Ch R = 1 ,3924    ,133.1,137.3,139.1
XS GIS Cut Line= 4
 2269525.9493696614592.0125097952269397.82305443614622.165475101
2269347.87700767614680.6772003972269269.68920689614733.531134939
#Sta/Elev= 30
       0    2440    14.2 2431.81      39 2415.33    52.3 2406.92    63.5 2401.01
    79.9 2391.07    92.2  2382.7   108.7 2370.22   116.9 2364.73   125.1  2358.4
   129.2 2355.78   135.6 2352.87   149.1  2350.3   152.6 2350.19     165 2351.89
     169 2351.53   177.7 2349.22  187.562344.851   198.7 2343.53   201.9 2343.99
     204 2344.85     213 2351.64   227.5 2359.68   232.3 2363.14   237.5 2365.68
   256.5  2379.3   280.9 2395.04     288 2400.65     295 2405.07   302.9 2410.88
#Mann= 3, -1 ,  0
       0     0.1       0  187.56   0.045       0     204     0.1       0
Bank Sta=187.56,204
XS Rating Curve= 0 ,0
Exp/Cntr=0.3,0.1

Type RM Length L Ch R = 1 ,3786    ,106.7,104.3,102.1
XS GIS Cut Line= 4
2269452.19887277614507.2803773292269304.66295592614548.407646186
2269272.50452216614566.088126939 2269210.0854876614629.209120544
#Sta/Elev= 30
       0  2414.5    29.1 2399.66    51.8 2384.36    76.2 2365.97    83.1 2361.69
    87.2  2359.6    96.4 2352.89   103.8 2348.47     108 2346.78   112.1 2346.07
   121.7 2346.31   131.5 2345.73   150.9 2347.95   153.7 2347.62     160 2343.22
  162.692342.106   176.5 2341.22  181.792342.104   185.7 2343.81   189.9 2348.18
     196 2352.76   201.7 2356.46   211.1  2360.9   222.3 2367.08   235.8 2375.63
   244.8 2382.16   258.6 2391.19   265.8 2397.04     273 2402.16   278.6 2406.99
#Mann= 3, -1 ,  0
       0     0.1       0  162.69   0.045       0  181.79     0.1       0
Bank Sta=162.69,181.79
XS Rating Curve= 0 ,0
Exp/Cntr(USF)=0,0
Exp/Cntr=0.3,0.1

Type RM Length L Ch R = 1 ,3682    ,121.2,128.9,135
XS GIS Cut Line= 4
2269371.81597528614398.2925440942269240.52309136614461.133139302
2269207.44427288614490.9070212732269148.77964697 614554.46033568
#Sta/Elev= 30
       0 2391.55    34.9  2376.1    52.8 2366.49    61.7  2362.7    66.1 2360.11
    79.4 2350.09    83.9 2347.92   101.6 2343.02   106.9 2343.12   114.9 2344.11
   123.8 2341.95   145.6 2341.71   151.4 2342.12   157.6  2343.4   162.2 2342.05
   167.6 2338.33  169.362337.771   172.9 2337.05   178.3 2336.85   181.5 2337.03
  183.492337.771   188.3  2340.3   193.2 2346.56   198.6 2351.37   206.7 2356.27
   220.4 2366.44   236.4 2379.76   253.4    2393   263.9 2399.82   276.6 2406.69
#Mann= 3, -1 ,  0
       0     0.1       0  169.36   0.045       0  183.49     0.1       0
Bank Sta=169.36,183.49
XS Rating Curve= 0 ,0
Exp/Cntr=0.3,0.1

Type RM Length L Ch R = 1 ,3553    ,109.2,108.7,107.7
XS GIS Cut Line= 4
2269329.43429981 614331.124763542269200.76470152614370.489435161
2269119.68522863614361.6764489772269043.30601504614431.005273623
#Sta/Elev= 30
       0 2386.28     9.7 2381.16    20.7  2376.7      39 2365.67      48 2359.41
    59.9 2353.74    72.4 2346.44    85.9 2341.48    89.2 2340.56    95.5 2340.35
   110.1  2343.5   114.8 2343.97   147.2  2337.6   151.2 2336.65   159.3 2333.84
   167.3 2333.23   175.4 2333.39  177.13 2333.81   179.4  2334.5   183.5 2337.84
   187.5 2342.71   191.5 2344.46   203.6 2344.22   215.6    2345   223.9 2346.59
   237.1  2350.9   242.5 2353.72   268.9 2369.26   286.2 2378.12   319.3  2392.7
#Mann= 3, -1 ,  0
       0     0.1       0   159.3   0.045       0  177.13     0.1       0
Bank Sta=159.3,177.13
XS Rating Curve= 0 ,0
Exp/Cntr(USF)=0,0
Exp/Cntr=0.3,0.1

Type RM Length L Ch R = 1 ,3444    ,119.7,118.6,115.2
XS GIS Cut Line= 4
2269320.17969089614252.4424876872269202.47081378614260.082722219
2269128.90189015614258.4963847062268992.27401604614341.460289266
#Sta/Elev= 30
       0 2388.17      16 2378.69    28.1 2369.15    36.1 2363.33    59.2 2348.04
    68.1  2343.1    80.2 2338.76   100.2 2335.37   108.2 2335.82   116.2 2338.37
   120.3 2337.94   124.3  2335.9   132.3 2330.92   136.3 2329.66   140.3 2329.59
  150.11 2330.93   152.3 2331.48   160.3 2336.24   164.3 2337.87   172.3 2339.02
   201.8 2340.46   239.2  2341.5   257.9 2342.43   262.6 2343.23   278.5 2349.04
   290.7 2355.28   304.7 2360.54   313.4 2366.16     328 2373.93   351.4  2387.6
#Mann= 5, -1 ,  0
       0     0.1       0   132.3   0.045       0  150.11     0.1       0
  177.96    0.05       0  251.54     0.1       0
Bank Sta=132.3,150.11
XS Rating Curve= 0 ,0
Exp/Cntr=0.3,0.1

Type RM Length L Ch R = 1 ,3326    ,138.1,131.1,121.4
XS GIS Cut Line= 4
2269294.33258141614117.9695738242269224.41622435614143.233467551
2269162.54906134614150.8478876142268976.47167106614262.208781033
#Sta/Elev= 30
       0  2400.3     6.5  2395.2    23.6 2384.29    32.1 2378.31    49.1 2365.34
    61.8 2354.81    66.7 2351.34    70.3 2347.84    74.3 2341.94    82.6  2331.5
    86.7 2326.69   88.13 2325.87    90.7 2325.22    98.8 2324.81   110.9 2325.83
   122.9 2328.44   137.2 2334.26   139.4 2334.83   144.1  2334.5   148.8 2334.98
   153.4 2337.24   157.6 2337.98   172.2 2336.78   215.9 2338.45   260.6 2338.04
   274.3 2339.15   293.3 2343.84   320.4 2355.02   339.9 2363.79   353.5 2370.57
#Mann= 5, -1 ,  0
       0     0.1       0   88.13   0.045       0   110.9     0.1       0
  166.67    0.05       0  276.67     0.1       0
Bank Sta=88.13,110.9
XS Rating Curve= 0 ,0
Exp/Cntr(USF)=0,0
Exp/Cntr=0.3,0.1

Type RM Length L Ch R = 1 ,3195    ,107.2,107.5,107.4
XS GIS Cut Line= 4
2269188.05069899613999.1456356072269127.65885438614035.027875255
2269062.62212568614113.4020466462268937.17049031614186.813948306
#Sta/Elev= 30
       0 2376.62     4.5 2373.68     9.2 2372.57    13.1 2370.84    18.5 2366.82
    33.5 2357.07    43.1 2349.98    58.8 2340.08      73 2329.14    79.9 2325.39
   84.992323.285    88.6  2322.4    93.8 2322.35      99 2322.57  101.352323.284
   104.2 2324.77   109.4 2329.16     114 2330.69     125 2330.42   132.1 2332.52
   135.4 2332.89   161.4 2332.58   198.1 2334.03   235.2 2337.42   243.9 2338.91
   257.8 2342.17   276.9 2348.68   284.8 2351.65   302.4  2359.7   317.4 2365.21
#Mann= 5, -1 ,  0
       0     0.1       0   84.99   0.045       0  101.35     0.1       0
  140.25    0.05       0  202.09     0.1       0
Bank Sta=84.99,101.35
XS Rating Curve= 0 ,0
Exp/Cntr=0.3,0.1

Type RM Length L Ch R = 1 ,3087    ,158.4,164.4,167.3
XS GIS Cut Line= 4
2269150.18185563613937.8614255022269043.89724225613969.059396592
2268985.73153344614037.8006888262268890.55128266614118.175122822
#Sta/Elev= 30
       0 2365.59    49.4 2344.25    52.6  2343.1    60.5  2341.9    65.5 2340.58
    81.3 2333.62    85.5 2332.23    97.8  2329.5   106.3 2327.17   110.6 2325.53
   116.3 2322.53  121.232321.096   130.5 2320.05   135.1 2320.34  138.062321.096
   147.5  2324.7   153.2    2324   156.1 2324.49   158.1 2325.19   163.3 2328.07
   172.3  2328.5     179 2331.03   181.6 2331.59   208.1  2332.8   218.6 2333.69
   244.7 2339.04   275.3 2344.68   289.5 2348.68   311.4  2357.2   325.4  2362.1
#Mann= 3, -1 ,  0
       0     0.1       0  121.23   0.045       0  138.06     0.1       0
Bank Sta=121.23,138.06
XS Rating Curve= 0 ,0
Exp/Cntr(USF)=0,0
Exp/Cntr=0.3,0.1

Type RM Length L Ch R = 1 ,2923    ,96.5,103.2,106.6
XS GIS Cut Line= 4
2269120.75521485613824.6253997582268945.70490836613863.766702685
2268906.97648437613879.951603194  2268819.082814613922.067589009
#Sta/Elev= 30
       0 2366.32     4.7 2364.64     8.8  2361.9    12.9 2359.83    34.4  2350.3
    41.6 2347.69    49.8 2343.39    53.9 2341.76    62.1 2337.67    66.2 2335.55
    70.3 2332.77    74.4 2330.91    94.9 2327.91   111.3 2326.13   127.7 2325.45
     140 2323.78   181.6 2321.17   185.4 2320.32   190.8 2317.43   196.72316.328
   203.8 2315.79  216.04 2316.32   228.9 2321.02   237.8 2328.85   242.2 2331.97
   248.4 2335.53   255.5 2340.28   278.3 2353.69     289 2359.32   318.8 2376.12
#Mann= 5, -1 ,  0
       0     0.1       0  179.37    0.06       0   196.7   0.045       0
  216.04    0.06       0  251.35     0.1       0
Bank Sta=196.7,216.04
XS Rating Curve= 0 ,0
Exp/Cntr=0.3,0.1

Type RM Length L Ch R = 1 ,2820    ,122,118.7,116.7
XS GIS Cut Line= 4
2269096.91510276613753.0799580662268954.60169624613777.234068348
2268869.73590336613766.7890476862268786.17573806613807.916316543
#Sta/Elev= 30
       0 2362.61    25.1 2350.27    41.3 2343.66    49.4 2339.41    53.5 2337.98
    61.6 2336.89    69.7 2333.69    81.9 2330.25    94.1 2326.23   104.8 2324.43
   114.4 2324.11   142.9 2320.43   146.8 2319.46   150.8 2317.66   154.9 2314.83
  158.772312.867   162.9  2312.4     175 2312.17   183.42312.867   191.1 2316.58
   195.2 2317.22   203.2 2317.16   215.3 2316.17   221.9 2316.07   231.6 2316.25
   236.1 2317.19   241.8 2319.64   262.4 2332.21   301.5 2353.08     323 2365.26
#Mann= 5, -1 ,  0
       0     0.1       0  154.35    0.06       0  158.77   0.045       0
   183.4    0.06       0  259.85     0.1       0
Bank Sta=158.77,183.4
XS Rating Curve= 0 ,0
Exp/Cntr(USF)=0,0
Exp/Cntr=0.3,0.1

Type RM Length L Ch R = 1 ,2701    ,105.1,103.7,102.9
XS GIS Cut Line= 4
2269100.44751638 613629.48060341 2268976.2866262613650.548984284
2268867.40668061613663.1482633492268736.37211007613724.479340057
#Sta/Elev= 30
       0  2380.3    24.3 2368.66    40.8 2360.02    57.1 2352.86    69.3 2345.32
    73.3 2343.68    81.4 2343.12    85.5 2341.36    93.8 2335.15   117.9 2322.51
   125.9 2319.65   134.1 2318.07   142.8 2313.83   150.2 2311.69  154.922308.615
   158.3 2307.47  177.062308.614   182.4 2309.59   190.5 2313.35   194.5 2314.31
   218.7 2315.06   239.1 2313.48   247.9 2313.45   260.6 2314.34   274.4 2316.91
   287.7 2317.85   296.2 2319.59   305.4 2322.85   332.8  2336.9   380.2 2364.06
#Mann= 4, -1 ,  0
       0     0.1       0  154.92   0.045       0  177.06    0.06       0
  265.54     0.1       0
Bank Sta=154.92,177.06
XS Rating Curve= 0 ,0
Exp/Cntr=0.3,0.1

Type RM Length L Ch R = 1 ,2597    ,127.1,126.5,126.9
XS GIS Cut Line= 4
2269077.96466164 613514.15382575 2268951.9715999613546.141701529
2268842.95169674613568.3373704362268702.59673159613632.965935784
#Sta/Elev= 30
       0 2387.17      37 2366.66    51.4 2359.65    55.5 2356.98    63.8 2349.44
    67.9 2347.94      72 2347.99    76.1 2346.61    86.2 2336.56   109.1  2320.9
   121.5 2316.01   125.7 2315.23   137.9 2315.08     142    2314  161.582303.955
   170.6 2302.75  179.562303.954   182.8 2305.51   186.9 2309.29     191 2311.42
   215.5 2312.34   257.5 2312.17   279.5 2314.61   301.6 2315.54   310.4 2317.16
   319.4 2319.53   336.8 2326.84   345.6 2329.45   376.4 2341.72   395.8  2350.5
#Mann= 5, -1 ,  0
       0     0.1       0  139.99    0.06       0  161.58   0.045       0
  179.56    0.06       0  311.25     0.1       0
Bank Sta=161.58,179.56
XS Rating Curve= 0 ,0
Exp/Cntr(USF)=0,0
Exp/Cntr=0.3,0.1

Type RM Length L Ch R = 1 ,2471    ,109.6,108.7,108.4
XS GIS Cut Line= 4
2269024.12136602613404.2032765482268910.39006673613425.254680002
2268844.74364469613439.6955966922268692.16665704613448.601528879
#Sta/Elev= 30
       0 2371.75       4 2368.44     8.1 2365.77    16.2 2364.38    24.4 2358.99
    28.3 2357.19    36.6 2350.72    48.8 2348.12    52.3 2346.05      61 2339.77
    77.2 2330.57    93.5 2322.12   105.7 2314.88   113.8 2308.96   117.9 2304.52
  121.562301.348     122    2301   127.5 2300.62   134.2 2300.69  138.832301.348
   146.6  2307.4   150.7 2308.66   175.3  2308.8   195.5  2307.8   211.7 2308.79
   235.5 2309.38   263.6 2311.97   315.7 2323.53   327.7 2327.19   335.7 2330.63
#Mann= 5, -1 ,  0
       0     0.1       0  121.56   0.045       0  138.83     0.1       0
  182.88    0.06       0  282.88     0.1       0
Bank Sta=121.56,138.83
XS Rating Curve= 0 ,0
Exp/Cntr=0.3,0.1

Type RM Length L Ch R = 1 ,2362    ,136.4,137.3,138.9
XS GIS Cut Line= 4
  2269011.205659613312.2600818612268890.07243327613316.612173804
2268794.32641053613344.9007714312268691.32690122613345.626120088
#Sta/Elev= 30
       0 2371.49    38.6 2351.63    47.1 2348.05    55.1 2342.05    63.1 2340.91
    95.1 2324.77   104.3 2319.62   114.3  2312.4   119.7  2307.8   126.4 2303.38
   135.7 2301.03  141.912298.551   148.2 2297.48  159.112298.552   160.7 2298.95
   164.9 2302.06   169.1 2304.26   177.4 2304.55   185.8 2302.58   189.9  2302.3
   210.8 2302.64   227.2 2305.29   243.2 2305.81   263.2 2309.97   275.1 2311.58
   283.4 2314.69   291.2 2319.68   303.2 2321.46   307.2  2322.8   324.1 2331.13
#Mann= 5, -1 ,  0
       0     0.1       0  141.91   0.045       0  159.11     0.1       0
  171.21    0.06       0  271.05     0.1       0
Bank Sta=141.91,159.11
XS Rating Curve= 0 ,0
Exp/Cntr(USF)=0,0
Exp/Cntr=0.3,0.1

Type RM Length L Ch R = 1 ,2225    ,119.5,117.9,116.1
XS GIS Cut Line= 4
2268978.27610165613225.3870026942268867.95273562613186.941529097
2268795.32254196613196.3420435132268679.88272762613223.306278522
#Sta/Elev= 30
       0 2355.58    23.4 2346.71    48.9  2334.7    61.5 2330.81    67.8 2327.35
    86.9 2319.02   108.1  2313.2   116.6 2310.17   120.6 2307.55   128.7 2301.09
   132.7  2298.9  147.97 2295.35   152.9 2294.46     161 2294.66  164.072295.351
   165.1 2295.59     169 2298.66   173.1 2300.77   177.1 2301.43   217.9 2301.32
   234.4 2302.68   238.5 2303.94   250.8 2312.09     260 2313.31   263.1 2314.59
   267.2 2317.37   291.9 2328.19     296 2330.56   304.2 2337.17   308.6 2339.26
#Mann= 5, -1 ,  0
       0     0.1       0  146.83    0.06       0  147.97   0.045       0
  164.07    0.06       0  240.07     0.1       0
Bank Sta=147.97,164.07
XS Rating Curve= 0 ,0
Exp/Cntr=0.3,0.1

Type RM Length L Ch R = 1 ,2107    ,126.3,125.9,124.5
XS GIS Cut Line= 4
2268934.51203961613009.2674464022268843.84345747613063.668595685
2268735.04115891613101.3867258542268655.97815528613118.795093625
#Sta/Elev= 30
       0 2362.14    23.2 2351.32    45.4 2339.82      82 2318.91      96 2311.99
   105.4 2306.06   110.3 2303.51   113.9  2301.8   122.3 2299.99   126.6 2297.59
   131.8 2293.29     135 2291.53   137.12290.886   143.5 2289.67   147.7 2289.55
     152 2289.97   153.62290.887   160.4 2294.91   164.7 2295.88   177.4 2296.33
   190.1 2297.66   211.2 2297.85   223.8 2300.58     232 2304.29   245.9 2312.92
   252.5 2316.44   260.7 2319.28   277.1  2322.1   280.2  2323.1   301.8 2332.61
#Mann= 5, -1 ,  0
       0     0.1       0  105.74    0.06       0   137.1   0.045       0
   153.6    0.06       0  230.89     0.1       0
Bank Sta=137.1,153.6
XS Rating Curve= 0 ,0
Exp/Cntr(USF)=0,0
Exp/Cntr=0.3,0.1

Type RM Length L Ch R = 1 ,1981    ,104.2,107.1,109.4
XS GIS Cut Line= 4
2268889.69301687612932.3572249012268804.73235005612947.518286945
2268718.44174434612979.2591629732268630.83277747613029.411927508
#Sta/Elev= 30
       0 2344.72    17.8 2333.42      30 2327.38    42.2 2319.73    70.6 2304.39
    78.7 2299.27    91.2 2289.44      942288.546   100.5 2287.68  116.822288.547
     121  2289.9   129.5 2291.33   134.8 2291.41   142.3 2290.68   155.1 2291.91
   163.6 2292.06   176.4 2294.68   180.9 2295.14   204.8 2294.42   213.6 2293.61
   217.7 2293.84   225.3 2297.45   231.6 2301.51   234.1 2303.56   248.7 2317.11
   259.2 2328.19   266.3 2334.13   269.2  2336.2   272.2 2337.58   279.2 2339.02
#Mann= 5, -1 ,  0
       0     0.1       0      94   0.045       0  116.82     0.1       0
   146.3    0.06       0  258.25     0.1       0
Bank Sta=94,116.82
XS Rating Curve= 0 ,0
Exp/Cntr=0.3,0.1

Type RM Length L Ch R = 1 ,1874    ,135.7,133,129.9
XS GIS Cut Line= 4
2268893.98996188612823.3356395392268796.45958145612846.249403617
2268723.42213471612855.5940478812268611.38687159612876.801089055
#Sta/Elev= 30
       0 2359.67    18.3 2349.05    26.5 2344.92    34.7 2340.02    38.8 2338.23
    47.1 2333.17    55.3 2328.74    82.9 2311.56    92.3 2304.12   104.5 2289.83
   108.5 2285.47  109.382285.056   112.6 2283.64  132.082285.055   136.8 2286.14
   140.8 2288.23   148.9 2290.43   152.9 2290.98     165 2290.29   185.3 2289.98
   197.5 2289.39   213.8 2289.62   222.5 2290.36   229.3  2292.3   234.1  2294.8
   242.3 2300.24   254.5    2311   273.8 2331.77   280.6 2339.85   287.8 2347.75
#Mann= 4, -1 ,  0
       0     0.1       0  109.38   0.045       0  132.08     0.1       0
  253.82    0.06       0
Bank Sta=109.38,132.08
XS Rating Curve= 0 ,0
Exp/Cntr(USF)=0,0
Exp/Cntr=0.3,0.1

Type RM Length L Ch R = 1 ,1741    ,118.4,119.1,120
XS GIS Cut Line= 4
2268846.90097537612693.9377583032268757.12907702612714.645391822
2268716.91886197 612731.860005882268600.73485399 612753.90448308
#Sta/Elev= 30
       0 2354.53      15 2346.23    38.3 2332.04    51.7 2322.98    72.6 2307.57
    80.8 2300.18    84.9 2295.84    93.2 2283.39   96.182281.963    97.5 2281.43
   106.2 2281.13   114.9 2281.62  115.762281.964   119.2 2282.78   123.6 2285.39
     128 2286.68   140.7 2286.24   152.9 2286.36   165.1  2285.5   173.3 2285.44
   181.4 2285.65   185.5 2286.37   189.6 2288.62   193.6 2291.69   197.7 2295.17
   205.8 2302.66   209.9    2306   216.3 2311.72   234.3 2326.52   254.1 2340.72
#Mann= 4, -1 ,  0
       0     0.1       0   96.18   0.045       0  115.76     0.1       0
  205.87    0.06       0
Bank Sta=96.18,115.76
XS Rating Curve= 0 ,0
Exp/Cntr=0.3,0.1
